HEC-RAS study MILLCK.prj: MILLCK

--- MILLCK.g01 (geometry) --- (continued)

Type RM Length L Ch R = 1 ,14934   ,208.5,209.3,209.8
XS GIS Cut Line= 3
2023835.93981051 305057.27531557  2023738.200523304958.159418377
2023663.86360011304883.822495483
#Sta/Elev= 30
       0  1894.7      10 1894.91    19.4 1894.59    25.7 1893.73    31.8 1891.65
    41.1 1885.99    50.4 1879.37    53.3 1877.75    57.3 1876.53    64.3 1874.96
    68.9 1874.67    76.4 1874.95    80.1  1876.1      81 1876.73    85.6 1881.33
    87.5 1882.55    89.8 1883.45   117.8  1884.5   131.6 1884.47   136.3 1884.82
   143.2  1886.2   150.1 1886.47   161.7 1887.26   164.1 1887.66   168.7 1889.16
     171 1889.41   182.6 1889.78   210.5 1891.81     229 1898.81244.3293  1906.5
#Mann= 5 ,-1 , 0
       0    .016       0    19.4      .1       0    57.3    .045       0
      81     .05       0   150.1      .1       0
Bank Sta=57.3,81
XS Rating Curve= 0 ,0
Exp/Cntr(USF)=0,0
Exp/Cntr=0.3,0.1

Type RM Length L Ch R = 1 ,14725   ,182,182.9,184.9
XS GIS Cut Line= 2
2023973.60077883304918.2377375642023807.03100716304725.512381912
#Sta/Elev= 30
       0 1890.61     9.5 1890.93    12.3 1890.71    15.6 1889.99    20.6 1888.02
    35.6 1878.55    40.7 1875.75    45.7 1874.01    50.7 1873.05    56.5 1872.49
    74.6 1872.01    83.2 1870.97    91.4 1868.81    96.1 1868.39   100.7  1867.5
   104.9 1867.32   110.9 1867.69   114.7 1868.71   117.9 1870.48   121.6  1873.7
   126.3 1877.26   130.9 1879.52     136 1881.04   156.9 1883.06   191.4 1884.67
   221.3  1884.8   239.3 1883.74   241.4 1884.09     248 1886.76254.7323    1889
#Mann= 4 ,-1 , 0
       0    .016       0    12.3      .1       0    96.1    .045       0
   114.7     .05       0
#Block Obstruct= 3 ,-1
  162.81  198.76  1904.7  207.59  216.38 1904.87  226.59  244.43 1905.34
Bank Sta=96.1,114.7
XS Rating Curve= 0 ,0
Exp/Cntr(USF)=0,0
Exp/Cntr=0.3,0.1

Type RM Length L Ch R = 1 ,14542   ,114.6,108.1,101.3
XS GIS Cut Line= 3
2024119.52140526304827.3814984712024054.82075014304748.914746527
2023897.88724626304618.136826621
#Sta/Elev= 30
       0 1887.51    19.1 1887.56    23.6  1887.3    30.5 1884.43    36.1 1882.55
    39.1 1880.91    46.8 1875.15    63.1 1862.22    65.9  1860.7    70.2 1859.78
    74.8 1859.93    77.1 1860.58    80.4 1862.37    84.1 1864.37    86.4 1865.01
    88.8 1865.22    95.7 1865.12   109.6  1862.8   114.9 1862.71   152.4 1864.98
   184.3 1867.66   214.5 1869.37   237.8 1869.47   248.2 1869.96   263.6 1870.04
   267.7 1870.58   272.8 1872.01   280.5 1874.24     289 1878.59305.9832 1884.89
#Mann= 5 ,-1 , 0
       0    .016       0    19.1      .1       0    63.1    .045       0
    80.4     .05       0   272.8      .1       0
#XS Ineff= 2 , 0
                           92.28            1867
Permanent Ineff=
       F       F
Bank Sta=63.1,80.4
XS Rating Curve= 0 ,0
Exp/Cntr(USF)=0,0
Exp/Cntr=0.5,0.3

Type RM Length L Ch R = 1 ,14434   ,38,38.5,39
XS GIS Cut Line= 3
2024237.80269266304723.1800975472024093.29171455304668.988480757
2023898.60331349304602.754282459
#Sta/Elev= 30
       0 1884.42    13.7  1884.4    21.3 1883.75    25.6 1882.78    30.3 1880.77
    53.6 1866.36    61.8 1861.97    65.3 1860.74    72.3 1859.22    79.9 1858.52
      91 1858.78   100.3 1859.62   103.8 1858.64   107.3 1856.59   109.7 1855.76
   115.6 1854.93   117.9 1854.98   121.4 1855.86   128.4 1860.41   131.9 1861.32
   156.3  1861.9   177.3 1863.95   215.3 1866.63   254.7 1867.88   296.1 1868.19
   301.9 1868.88   319.1  1873.4   329.6 1879.11   339.9 1883.25359.9844 1888.98
#Mann= 5 ,-1 , 0
       0    .016       0    21.3      .1       0   109.7    .045       0
   121.4     .05       0   301.9      .1       0
#XS Ineff= 3 ,-1
       0      88    1864      88      99 1858.73     131     200  1861.7
Permanent Ineff=
       F       F       F
#Block Obstruct= 1 ,-1
  231.51  262.38 1887.82
Bank Sta=109.7,121.4
XS Rating Curve= 0 ,0
Exp/Cntr(USF)=0,0
Exp/Cntr=0.5,0.3

Type RM Length L Ch R = 2 ,14421   ,,,
BEGIN DESCRIPTION:
Private Driveway
Survey ID: MIC020
END DESCRIPTION:
Bridge Culvert--1,0,-1,-1, 0
Deck Dist Width WeirC Skew NumUp NumDn MinLoCord MaxHiCord MaxSubmerge Is_Ogee
11,12,2.6,0, 5, 5, , , 0.98, 0, 0,0,,
      85     100     116     130     170
    18581860.3691860.8511860.9941860.994
                                        
      85     114     128     144     170
    18581860.3691860.8511860.9941860.994
                                        
BR Coef=-1 , 1 , 0 ,, 0 ,,,0.8,0,1.2,0,
WSPro=,,,, 1 ,,,, 0 ,,,, 0 ,,,,-1 ,-1 ,-1 , 0 , 0 , 0 , 0 , 0
Culvert=2,6,10,12,0.012,0.2,1,8,1,1854.234,115,1853.849,128,Culvert #1  , 0 ,11
     115     128
BC Culvert Barrel=1,Barrel1,0
Culvert Bottom n=0.012
BC Design=,, 0 ,, 0 ,,,,,,
BC Use User HTab Curves=0
BC User HTab FreeFlow(D)= 0

Type RM Length L Ch R = 1 ,14396   ,142.2,145.1,144.8
XS GIS Cut Line= 4
2024265.90204951304697.0878376112024167.55430052304656.945899249
2024111.35558682304632.8607362312023940.75234877304573.651377146
#Sta/Elev= 30
       0 1883.57      10 1883.29    15.1 1882.82    20.1 1881.48    25.5 1879.57
    36.1 1874.02    47.8 1866.31    55.3 1860.76    58.9 1859.15    65.4 1858.46
   110.7 1858.22   114.2 1857.54   121.3 1853.82   125.6 1852.98     132 1853.31
   135.6  1854.6   139.1 1856.69   142.7 1858.35   145.6 1858.86   171.2 1860.68
   188.5 1862.41   199.1 1863.08   237.1 1866.44     258 1867.06   282.3  1866.5
   289.3 1866.04   292.7 1866.29   310.1 1870.11     321 1875.77347.9527 1887.68
#Mann= 3 ,-1 , 0
       0      .1       0   121.3    .045       0   135.6     .05       0
#XS Ineff= 2 , 0
       0     116  1856.2     141       0    1861
Permanent Ineff=
       F       F
#Block Obstruct= 1 ,-1
  230.52  261.38  1886.9
Bank Sta=121.3,135.6
XS Rating Curve= 0 ,0
Exp/Cntr(USF)=0,0
Exp/Cntr=0.5,0.3

Type RM Length L Ch R = 1 ,14250   ,203.7,207.2,210.3
XS GIS Cut Line= 2
2024342.53217394304598.8642910562024118.14479557304465.333151783
#Sta/Elev= 30
       0 1873.28     2.1 1872.52     5.4 1871.84    18.3 1870.78    22.5 1869.09
    40.3 1859.81    44.1 1858.36    55.6 1855.62      68 1853.68    74.7 1853.15
    86.1    1853    97.6 1853.38     109 1851.32   116.7 1850.51     123  1848.7
   127.8 1847.77   137.4 1847.68   139.8 1847.71   144.6 1848.75   154.8 1853.16
   161.3 1854.12   187.7 1855.16   192.4 1854.88   197.9 1853.95   208.3 1853.53
   216.4 1854.66   223.5 1856.93   231.2 1858.97   254.7 1866.93261.1135  1869.5
#Mann= 3 ,-1 , 0
       0     .05       0     123    .045       0   144.6      .1       0
Bank Sta=123,144.6
XS Rating Curve= 0 ,0
Exp/Cntr(USF)=0,0
Exp/Cntr=0.3,0.1

Type RM Length L Ch R = 1 ,14043   ,229,226.9,220.5
XS GIS Cut Line= 2
2024466.42704543304457.0734936832024261.31220263304294.633551063
#Sta/Elev= 30
       0 1877.25    18.6 1876.39    22.3 1875.95    24.5 1875.19    27.9 1873.15
    41.9 1861.18    45.6 1858.55    53.6 1853.96    59.9 1851.69    64.1 1850.59
    76.9 1848.54   100.3 1847.64     106  1846.2   116.7 1841.55   122.7 1839.91
   128.3 1839.25   131.1 1839.33   137.7    1841     146 1842.99     154 1843.31
   161.9 1844.49   189.1  1844.3   196.1 1845.05   202.2  1846.3   206.4 1847.54
   210.6 1849.39   223.1 1856.65   235.8  1863.4   247.4 1867.59261.6464 1871.57
#Mann= 3 ,-1 , 0
       0     .05       0   116.7    .045       0   137.7      .1       0
#XS Ineff= 2 , 0
                          163.44         1845.57
Permanent Ineff=
       F       F
#Block Obstruct= 1 ,-1
   13.26   26.57 1896.71
Bank Sta=116.7,137.7
XS Rating Curve= 0 ,0
Exp/Cntr(USF)=0,0
Exp/Cntr=0.3,0.1

Type RM Length L Ch R = 1 ,13816   ,187.3,187.1,186.5
XS GIS Cut Line= 2
2024637.12664615304260.2183089822024396.21995158304147.336314958
#Sta/Elev= 30
       0 1861.75     4.9 1861.81    12.1 1861.32    30.2 1858.97    41.1 1857.92
    55.6 1857.29      81 1855.32   106.3  1854.1     110 1852.37   113.4 1849.45
   117.2 1847.49   124.4  1846.4   128.1 1845.24   135.6 1840.28   142.6 1836.01
   146.2 1834.14   150.4 1833.05   153.4 1832.66   157.1 1832.61   160.7 1833.26
   164.3 1834.48   167.9 1835.33   175.1 1835.69   189.7 1835.91   209.4 1837.58
   218.6 1838.12   240.4  1840.1   244.6 1840.81   251.3 1842.61266.0421 1847.34
#Mann= 3 ,-1 , 0
       0     .05       0   146.2    .045       0   164.3      .1       0
#Block Obstruct= 2 ,-1
   51.03   84.33 1877.54   98.94  132.77 1874.56
Bank Sta=146.2,164.3
XS Rating Curve= 0 ,0
Exp/Cntr(USF)=0,0
Exp/Cntr=0.3,0.1

Type RM Length L Ch R = 1 ,13629   ,81.4,86.8,89.7
XS GIS Cut Line= 2
2024718.34661746304092.2719276292024485.69958099303983.519762654
#Sta/Elev= 30
       0 1841.27     8.7 1841.23    80.9 1838.66    96.4 1837.69    98.2 1837.54
   100.1  1837.1     109 1834.36   114.9 1833.08   127.2 1831.81   141.6 1830.63
   148.9 1830.55   152.5 1829.33   154.3 1828.48   156.1 1827.77   156.8 1827.71
   176.6 1827.31   181.5  1827.5   185.1  1828.1   192.3 1829.12   203.2 1829.12
   206.8 1830.22   208.6 1831.78   210.4 1833.66     216 1842.57   218.5 1845.69
   221.3 1848.47   224.9 1851.16   238.3 1860.19   245.7  1865.4256.8106 1873.55
#Mann= 4 ,-1 , 0
       0     .05       0   100.1      .1       0   154.3    .045       0
   185.1      .1       0
#Block Obstruct= 2 ,-1
   47.48   61.79 1859.87   68.77   88.79 1859.11
Bank Sta=154.3,185.1
XS Rating Curve= 0 ,0
Exp/Cntr(USF)=0,0
Exp/Cntr=0.3,0.1

Type RM Length L Ch R = 1 ,13543   ,113.2,111,109.7
XS GIS Cut Line= 4
2024757.22225412304034.9198901952024628.85405114303963.381360408
2024606.12218186303945.3295818642024559.32127453303919.254790633
#Sta/Elev= 30
       0 1837.57       7 1837.52    44.9 1835.97    59.9 1835.01    74.9 1835.12
    79.4 1835.39    81.8 1835.41    84.2 1834.95    87.3 1833.87    93.8 1830.27
    98.7 1828.94   103.5 1828.17   108.3 1827.74   127.6 1827.41   137.3 1826.34
   150.4 1826.64   155.81826.055   160.9 1825.67   168.9 1826.21   172.6 1826.19
   180.4 1826.39   186.9 1824.98   190.6 1825.95   191.8 1826.77   195.1 1829.79
   198.1 1832.99   201.9 1836.64   205.6  1839.5   220.7 1850.54   229.6 1857.59
#Mann= 4 ,-1 , 0
       0     .05       0    79.4      .1       0   155.8    .045       0
   172.6      .1       0
#XS Ineff= 2 , 0
          126.76 1830.05
Permanent Ineff=
       F       F
#Block Obstruct= 1 ,-1
      31      51    1850
Bank Sta=155.8,172.6
XS Rating Curve= 0 ,0
Exp/Cntr(USF)=0,0
Exp/Cntr=0.3,0.1

Type RM Length L Ch R = 1 ,13432   ,147.5,146.9,145.9
XS GIS Cut Line= 2
2024828.47539212303946.3513012072024627.49037837303832.092697499
#Sta/Elev= 30
       0 1839.94      16 1837.01    35.2 1834.51    40.3 1833.25    55.4 1828.56
    59.1 1828.14    70.5 1827.54    90.5  1823.3    97.8 1821.28   100.7 1821.02
   115.8 1821.26   124.2 1822.74   134.6 1823.21     161 1822.52   164.8  1822.3
   167.5 1821.46   168.6 1821.06   172.4 1818.67   174.8 1817.53   176.1 1817.02
   179.6 1816.68   191.2 1817.15     195 1817.89   201.2  1820.3     206 1821.53
   208.4 1823.05   210.9 1825.16   217.6 1832.55   225.2 1838.84231.1926 1844.51
#Mann= 3 ,-1 , 0
       0      .1       0   174.8    .045       0     195      .1       0
#XS Ineff= 2 , 0
          136.62 1823.37
Permanent Ineff=
       F       F
Bank Sta=174.8,195
XS Rating Curve= 0 ,0
Exp/Cntr(USF)=0,0
Exp/Cntr=0.3,0.1

Type RM Length L Ch R = 1 ,13285   ,155.9,155.6,154.3
XS GIS Cut Line= 2
2024875.28012135303801.8072844682024707.33373999303710.951045375
#Sta/Elev= 30
       0 1826.36     3.5 1824.57     7.2 1823.08      11 1822.09    18.4 1821.23
    45.6  1819.9    61.4 1819.52    70.6 1819.11    81.9 1819.04      93  1819.3
   100.5 1818.87   102.8 1818.53   106.1 1817.82   111.7 1816.39   115.8 1814.73
   119.1 1813.63   126.6 1812.19   130.3 1811.78   135.2 1811.62   141.5 1811.66
     149 1812.12   149.7 1812.26   156.4 1813.85   160.2  1813.8   163.9 1814.04
   167.6 1814.95   171.4 1816.19   175.1 1817.88   181.2 1821.22190.9472  1827.3
#Mann= 3 ,-1 , 0
       0      .1       0   126.6    .045       0   149.7      .1       0
Bank Sta=126.6,149.7
XS Rating Curve= 0 ,0
Exp/Cntr(USF)=0,0
Exp/Cntr=0.3,0.1

Type RM Length L Ch R = 1 ,13129   ,228.9,229.5,228.5
XS GIS Cut Line= 2
2024946.86382487 303657.263267732024777.54083384303576.043296419
#Sta/Elev= 30
       0 1822.27     2.8 1822.06     6.4 1821.19     8.9 1819.88    13.8 1816.85
    16.2 1815.62    20.9  1813.9    24.6  1813.2    28.5 1812.78    53.7 1812.34
      61 1812.46    71.9 1813.17    75.3 1813.15    79.2 1813.02    86.4 1812.42
    90.1  1812.4   104.8 1813.33   108.3 1812.47   114.6 1810.08   122.8 1807.26
   126.5 1806.41   130.1 1806.21     141 1806.14   148.3  1806.9   150.6 1807.79
   151.9 1808.55   159.2    1816   161.3 1817.46   163.8    1819 187.795 1831.71
#Mann= 4 ,-1 , 0
       0     .05       0    75.3      .1       0   126.5    .045       0
   148.3      .1       0
Bank Sta=126.5,148.3
XS Rating Curve= 0 ,0
Exp/Cntr(USF)=0,0
Exp/Cntr=0.3,0.1

Type RM Length L Ch R = 1 ,12899   ,153.7,155.8,154.3
XS GIS Cut Line= 2
2025073.51191573303463.1613023952024851.87775673303364.045405203
#Sta/Elev= 30
       0 1814.46     8.5  1814.2    19.3  1810.6    22.9 1810.57      30 1811.46
    44.4 1811.49    55.2 1810.76    69.8 1810.05    80.4 1808.33    99.4 1806.04
   114.3 1803.44   119.9 1802.81   123.5 1801.75   127.1 1799.61   130.7 1798.19
   137.9 1796.77   141.5 1796.99     145 1798.09   148.6 1799.58   159.4 1800.24
   170.2 1802.27   191.8 1802.05   202.6 1802.92   206.4 1803.87   213.7 1807.12
   216.2 1808.58   220.5 1811.83   231.1 1821.01   238.4 1828.84242.7873 1833.12
#Mann= 5 ,-1 , 0
       0     .05       0      30    .016       0    55.2     .05       0
   130.7    .045       0     145      .1       0
#Block Obstruct= 1 ,-1
   91.65  123.86 1827.14
Bank Sta=130.7,145
XS Rating Curve= 0 ,0
Exp/Cntr(USF)=0,0
Exp/Cntr=0.3,0.1

Type RM Length L Ch R = 1 ,12744   ,236.4,234.1,231.3
XS GIS Cut Line= 2
2025183.64069039303339.2664309052024923.46146026303237.397314346
#Sta/Elev= 30
       0 1809.27     9.7 1809.54    22.4 1809.47    52.6  1808.5    59.6 1807.74
    66.7 1806.49    70.2 1806.06    84.3 1805.28    94.9 1805.36     106 1805.06
   133.6 1801.89     149 1799.41   159.1 1797.49   171.8  1796.6     183 1796.59
     197 1796.96   207.6 1796.66   211.1 1796.15   218.2 1794.08   221.7 1793.52
   225.2 1793.24   232.3 1793.14   242.8 1793.28   246.4 1794.05   250.3 1796.54
   256.9 1802.88   260.3 1805.41   267.5 1811.28   273.1 1815.55279.4111 1820.61
#Mann= 5 ,-1 , 0
       0     .05       0    84.3    .016       0     106     .05       0
   221.7    .045       0   246.4      .1       0
#XS Ineff= 2 , 0
          197.07 1798.34
Permanent Ineff=
       F       F
#Block Obstruct= 2 ,-1
    9.35   25.56 1829.53  184.07  195.01 1816.88
Bank Sta=221.7,246.4
XS Rating Curve= 0 ,0
Exp/Cntr(USF)=0,0
Exp/Cntr=0.3,0.1

Type RM Length L Ch R = 1 ,12510   ,153.3,154.1,151.3
Node Name=D
XS GIS Cut Line= 2
2025277.25014885303131.3983687372025047.35633175 303051.55500711
#Sta/Elev= 30
       0 1804.52    15.5 1801.88    36.3 1799.85    46.7 1798.11    71.1 1797.01
    82.5 1795.94    95.4 1796.13   119.7 1795.71   123.1 1795.26   126.6 1793.37
   134.1 1787.16     137 1786.16   140.5 1786.06   150.9 1787.66   155.6 1787.94
   162.5 1789.39   165.6 1789.42   170.2 1788.25   175.2 1787.36   177.9 1787.37
   185.7 1787.94   188.2 1788.53   192.6 1789.35   206.5 1790.03   223.9 1791.37
   227.3 1792.08   230.8 1793.49   234.3 1795.45   237.8 1798.27243.3642 1804.26
#Mann= 5 ,-1 , 0
       0     .05       0    95.4    .016       0   119.7     .05       0
   170.2    .045       0   188.2      .1       0
#Block Obstruct= 2 ,-1
    20.5   43.34 1821.37   46.84   64.15  1818.1
Bank Sta=170.2,188.2
XS Rating Curve= 0 ,0
Exp/Cntr(USF)=0,0
Exp/Cntr=0.3,0.1

Type RM Length L Ch R = 1 ,12355   ,166.9,165.3,164
XS GIS Cut Line= 2
2025317.17182966  302970.33503582025098.29089003302918.023867838
#Sta/Elev= 30
       0 1801.92    25.7  1798.3    29.1  1797.1    39.2  1792.9      46 1790.55
    49.3 1789.74    65.6 1789.01    73.8  1789.9    79.7 1789.97    92.8 1789.49
    99.9 1788.86   106.7 1787.41   123.5 1785.63   130.3 1783.54     137 1780.58
   139.1 1780.05   143.8 1779.14   147.2 1778.98   153.9 1779.19   160.3 1780.33
   167.4 1782.17   174.1 1783.59   177.5 1783.85   184.3 1783.65   187.6 1783.82
     191 1784.79   194.4 1786.61     218 1801.33   221.4 1802.65225.0452 1803.56
#Mann= 5 ,-1 , 0
       0     .05       0    73.8    .016       0    92.8     .05       0
   139.1    .045       0   160.3      .1       0
Bank Sta=139.1,160.3
XS Rating Curve= 0 ,0
Exp/Cntr(USF)=0,0
Exp/Cntr=0.3,0.1

Type RM Length L Ch R = 1 ,12190   ,202.9,203.9,204.9
XS GIS Cut Line= 2
2025392.88536224302798.2588253972025124.44647401302762.466973633
#Sta/Elev= 30
       0 1798.42     8.9 1797.11    22.6 1794.46      42  1791.6    71.8 1789.96
    75.1 1789.03    85.1 1783.26    88.4 1782.54    98.3 1783.14   121.5 1781.85
   131.4 1780.73   141.3    1780     148 1779.73   164.5  1779.7   177.8 1779.01
   181.1  1778.4   184.4 1776.72   187.7 1774.52     189  1774.1     191  1773.5
   203.6 1773.55   210.9 1773.06   214.2 1773.56   216.5 1774.46   224.1 1778.09
     234 1783.94   237.3  1786.2   250.8 1796.92     262 1804.36270.8145 1809.68
#Mann= 5 ,-1 , 0
       0     .05       0    98.3    .016       0   121.5     .05       0
     189    .045       0   216.5      .1       0
#Block Obstruct= 1 ,-1
  142.34   180.1 1799.95
Bank Sta=189,216.5
XS Rating Curve= 0 ,0
Exp/Cntr(USF)=0,0
Exp/Cntr=0.3,0.1

Type RM Length L Ch R = 1 ,11986   ,216.7,216,215.6
XS GIS Cut Line= 3
2025413.53450749302606.9100794292025167.12137419302561.481959882
 2025034.9668446302540.832814634
#Sta/Elev= 30
       0 1801.58     4.8 1799.01    16.7 1798.92      30 1793.64    33.4 1791.19
    42.1 1781.76      50 1777.74    70.1 1774.76    92.1 1775.14   106.7 1774.27
   189.4  1775.7   193.5 1774.64   200.2 1767.99     202 1766.96   203.5 1766.12
   213.9 1765.76   230.3 1767.24   240.2 1773.21   253.5 1773.74   260.2 1775.15
   263.5 1777.85   270.1 1785.88   273.4 1788.51   280.1 1792.64   286.1 1794.87
   313.7 1798.54   333.1  1805.1   347.5 1812.62   373.1 1815.17384.3237 1818.21
#Mann= 6 ,-1 , 0
       0    .016       0    16.7     .05       0    92.1    .016       0
   189.4     .05       0     202    .045       0   230.3      .1       0
#Block Obstruct= 1 ,-1
  350.29  378.35 1836.73
Bank Sta=202,230.3
XS Rating Curve= 0 ,0
Exp/Cntr(USF)=0,0
Exp/Cntr=0.3,0.1

Type RM Length L Ch R = 1 ,11770   ,219.5,219.4,220
XS GIS Cut Line= 3
2025454.83279798302386.6525301132025202.91322595302350.860678349
2025056.99259953302341.224410566
#Sta/Elev= 30
       0 1809.71    21.8 1807.88    38.4 1805.45    71.5 1797.37    74.8 1795.69
    78.2 1791.79    91.4 1771.03    94.7 1768.17      98 1766.84   104.9 1766.47
   117.9 1766.88   157.7 1766.09   184.2 1767.21   190.8    1767   197.5 1765.41
   208.7  1759.2     214 1757.26   223.1 1756.75   227.3 1757.41   230.6 1758.98
   237.2 1762.61   266.9 1762.32   283.4 1763.65   299.8 1763.94   306.4 1765.13
   319.6  1769.7     336 1780.69   345.9 1785.43   375.4 1793.66400.6879 1798.98
#Mann= 5 ,-1 , 0
       0      .1       0   104.9    .016       0   184.2      .1       0
   208.7    .045       0   230.6      .1       0
Bank Sta=208.7,230.6
XS Rating Curve= 0 ,0
Exp/Cntr(USF)=0,0
Exp/Cntr=0.3,0.1

Type RM Length L Ch R = 1 ,11551   ,201.2,199.4,196.2
XS GIS Cut Line= 3
 2025469.9755045302193.9271744612025249.71795518302137.486177449
2025098.29089003302114.083812834
#Sta/Elev= 30
       0 1809.73    41.3 1796.88    51.5 1792.37    61.6  1786.3      65 1782.11
    71.8 1771.62    79.1 1762.05      82    1760    95.5 1758.64   118.7 1759.23
   140.3  1758.3   146.3 1756.05   153.1 1750.52   163.2 1748.59     170 1748.78
   180.7 1750.88   191.5 1751.64   194.2 1752.44   200.5 1756.08     205 1757.22
   247.5 1757.46     261 1758.55   290.7 1759.16   300.6 1762.53   320.5 1771.88
     330 1773.86   343.8 1774.45   346.9 1775.68   353.7 1779.33380.5988 1790.62
#Mann= 7 ,-1 , 0
       0      .1       0    95.5    .016       0   118.7     .05       0
   153.1    .045       0   180.7      .1       0     330    .016       0
   346.9      .1       0
Bank Sta=153.1,180.7
XS Rating Curve= 0 ,0
Exp/Cntr(USF)=0,0
Exp/Cntr=0.3,0.1

Type RM Length L Ch R = 1 ,11351   ,209.3,230,243
XS GIS Cut Line= 3
2025474.10533355301975.0462348282025182.26408071301936.501163698
2025139.58918053301933.747944332
#Sta/Elev= 30
       0 1802.38    14.8 1798.83    47.9 1787.65    51.2 1784.01    64.4 1761.51
    67.7 1756.66      71 1753.68    80.9 1751.84    94.2 1752.32     114 1751.33
     124 1749.88   130.6  1746.7   140.5 1744.67   143.8 1742.83   150.4 1741.16
   157.1 1741.47   163.7 1743.11   184.4 1745.47   190.2 1747.25   199.6 1751.73
   203.4 1752.43   213.3 1751.93   226.7 1755.38   235.5 1756.75   256.3 1758.38
   266.3 1758.35     296 1761.38   305.9 1765.28   319.1 1768.63337.1393 1774.51
#Mann= 5 ,-1 , 0
       0      .1       0    94.2    .016       0     114     .05       0
   143.8    .045       0   163.7     .05       0
#Block Obstruct= 2 ,-1
     208     260 1778.26     267     287 1781.09
Bank Sta=143.8,163.7
XS Rating Curve= 0 ,0
Exp/Cntr(USF)=0,0
Exp/Cntr=0.5,0.3

Type RM Length L Ch R = 1 ,11121   ,99.8,92.1,89.1
XS GIS Cut Line= 6
2025458.43786098301950.7741741552025419.41097646301866.030082056
2025349.16258432301752.2945900282025314.59591518301706.577382448
2025238.77225383301675.3558748332025083.77976959301636.328990313
#Sta/Elev= 30
       0 1796.53    52.4 1789.21    57.9 1787.61    68.1 1784.16    87.5 1774.31
    92.9 1770.39   104.4 1758.96   110.7 1754.98   119.8 1750.81   128.3 1747.65
     133  1746.9   154.5 1747.19   218.8 1743.66     227 1742.15   240.2 1736.22
   250.8 1733.69   264.9 1733.09   272.6 1734.81   275.2 1736.62   281.3 1740.06
   294.4 1741.35   301.5 1744.86     305 1745.71   352.4 1745.76   382.3 1746.66
   389.1  1747.1   416.1 1751.89   429.7 1752.85   467.6  1761.5526.1244 1773.32
#Mann= 5 ,-1 , 0
       0      .1       0   154.5    .016       0   218.8     .05       0
   240.2    .045       0   275.2     .05       0
#XS Ineff= 2 , 0
             225 1743.59     289         1741.57
Permanent Ineff=
       F       F
#Block Obstruct= 3 ,-1
  300.84   324.1 1765.57  361.25     403 1765.99     407     420 1765.99
Bank Sta=240.2,275.2
XS Rating Curve= 0 ,0
Exp/Cntr(USF)=0,0
Exp/Cntr=0.5,0.3

Type RM Length L Ch R = 2 ,11083   ,,,
BEGIN DESCRIPTION:
Elton Lawn Road
Survey ID: MIC010
END DESCRIPTION:
Bridge Culvert--1,0,-1,-1, 0
Deck Dist Width WeirC Skew NumUp NumDn MinLoCord MaxHiCord MaxSubmerge Is_Ogee
16,50,2.6,0, 156, 6, , , 0.98, 0, 0,0,,
     180     222     245     258     284     296 296.279 296.279 296.513 296.816
 296.816 298.852  299.51  299.51 300.291 300.291 301.316 303.805 303.805 303.829
 303.839 303.839 303.863 306.342 307.387 307.387 308.856 309.895 310.935 310.935
 311.369 312.422 312.422 313.882 314.483 314.483 315.926 316.395 318.031 318.031
 318.909 321.039 321.039 321.422  321.58  321.58 321.958 323.935 325.128 325.128
 326.448  327.99 328.676 328.676 328.961 329.655 329.655 331.475 332.224 332.224
 333.988 334.022 335.772 335.772 336.501 338.272 338.272 339.014  339.32  339.32
 340.053 341.528 342.868 342.868 344.041 346.085 346.416 346.416 346.554 346.889
 346.889 349.067 349.964 349.964  351.58 352.117 353.512 353.512 354.094 355.506
 355.506 356.607  357.06  357.06 358.149  359.12 360.608 360.608 361.633 364.123
 364.123 364.147 364.156 364.156  364.18  366.66 367.705 367.705 369.173 370.212
 371.253 371.253 371.686 372.739 372.739 374.199 374.801 374.801 376.244 376.713
 378.349 378.349 379.226 381.356 381.356  381.51  381.51 381.747 381.887 381.887
 382.164 384.345 384.458 384.458 385.323 385.323 386.968 387.043 388.706 388.706
 389.746  391.49  392.09  392.09 392.448 393.872 393.872 395.151 395.473 395.473
 396.012 397.854 398.856 398.856 400.533 400.556
1743.5861743.5861743.3651743.0891742.1611741.4951740.5721740.5721740.5821740.586
1740.5861740.585 1740.58 1740.581740.5681740.5681740.5671740.5321740.5321740.531
1740.5311740.5311740.5311740.5181740.5131740.5131740.4921740.4781740.4631740.463
1740.4631740.4561740.4561740.4431740.4381740.4381740.4571740.464 1740.48 1740.48
 1740.551740.6541740.6541740.674 1740.68 1740.681740.6941740.801 1740.82 1740.82
1740.7961740.7291740.7061740.7061740.7131740.7251740.725 1740.82 1740.86 1740.86
1741.0761741.0811741.3091741.3091741.4071741.6561741.6561741.7491741.7821741.782
1741.8421741.9651742.0691742.0691742.1441742.2751742.2971742.2971742.308 1742.34
 1742.341742.5611742.6741742.6741742.9071742.9911743.2021743.2021743.2691743.433
1743.4331743.541 1743.58 1743.581743.6491743.7131743.8021743.8021743.8641743.997
1743.9971743.9981743.9991743.999    17441744.0841744.1331744.1331744.2341744.338
1744.4281744.4281744.4671744.5761744.5761744.7331744.7981744.7981744.8761744.902
1744.9911744.9911745.0271745.1281745.1281745.1351745.1351745.1461745.1531745.153
1745.1641745.2491745.2541745.254 1745.29 1745.291745.3581745.361 1745.43 1745.43
1745.4831745.5721745.6021745.6021745.6191745.6931745.6931745.7621745.7811745.781
1745.8161745.935    1746    17461746.1241746.126
                                                                                
                                                                                
                                                                                
                                                                                
                                                                                
                                                                                
                                                                                
                                                                                
                                                                                
                                                                                
                                                                                
                                                                                
                                                                                
                                                                                
                                                                                
                                                
     180     259     291     334     355     382
1743.5861743.5861743.3651743.0891742.1611741.495
                                                
BR Coef=-1 , 1 , 0 ,, 0 ,,,0.8,0,1.2,0,
WSPro=,,,, 1 ,,,, 0 ,,,, 0 ,,,,-1 ,-1 ,-1 , 0 , 0 , 0 , 0 , 0
Culvert=2,5,20,50,0.012,0.4,1,8,1,1732.993,257,1731.701,329,Culvert #1  , 0 ,15
     257     329
BC Culvert Barrel=1,Barrel1,0
Culvert Bottom n=0.012
BC Design=,, 0 ,, 0 ,,,,,,
BC Use User HTab Curves=0
BC User HTab FreeFlow(D)= 0

Type RM Length L Ch R = 1 ,11029   ,103.2,72,54.7
XS GIS Cut Line= 5
2025533.15387693301925.2682319372025426.10129952301695.426844014
 2025335.7819382301611.7978057582025189.70988472301578.346190456
2025068.16901578301572.770921239
#Sta/Elev= 30
       0 1794.09    39.6 1790.85    72.1 1785.02    90.2 1779.34    97.3 1772.83
   112.3 1763.54   119.2 1760.41   131.8 1758.14   144.2 1753.47   155.4 1747.59
     188 1746.25   213.3 1744.81   267.4 1743.86     302 1741.09   306.1 1739.83
   315.4 1733.48   317.9 1732.92   320.6 1731.89   325.4 1731.69   339.9 1732.46
   351.1 1737.86   364.6 1741.27   394.5 1741.06   411.4 1739.86   428.6 1737.41
     445 1736.88   455.1 1738.35   475.3 1743.79     539 1745.98   648.2    1766
#Mann= 5 ,-1 , 0
       0      .1       0   131.8    .016       0     188     .05       0
   317.9    .045       0   339.9     .05       0
#XS Ineff= 2 , 0
             303  1736.7     354         1735.85
Permanent Ineff=
       F       F
#Block Obstruct= 2 ,-1
  211.27  259.48 1765.05  423.33  479.52 1763.38
Bank Sta=317.9,339.9
XS Rating Curve= 0 ,0
Exp/Cntr(USF)=0,0
Exp/Cntr=0.5,0.3

Type RM Length L Ch R = 1 ,10957   ,117.1,113.5,113.8
XS GIS Cut Line= 5
2025504.29858737 301516.027636232025391.10660963301575.739759192
 2025330.2776606301588.7750190142025187.83123814301571.991967982
2025082.94457233301566.513375118
#Sta/Elev= 30
       0 1779.23    12.7 1773.75    26.7 1769.33    35.8 1765.08    43.3 1760.78
    54.4 1752.36    65.5 1745.23    72.9 1742.04    83.7 1740.61    86.1 1739.76
      90 1737.87   100.7 1730.62   106.3 1729.21   121.2 1728.78   138.6  1729.8
   148.7 1732.91   157.7 1732.69   165.4 1733.74   172.1 1733.79   175.5 1734.51
   185.6 1738.96   192.2 1740.33   208.8 1740.59   228.6 1739.38   248.4 1736.61
   264.9 1736.62   314.7 1743.67   347.4 1745.79   403.3 1755.32438.6477  1762.3
#Mann= 5 ,-1 , 0
       0      .1       0   100.7    .045       0   138.6      .1       0
   192.2    .016       0   228.6     .05       0
Bank Sta=100.7,138.6
XS Rating Curve= 0 ,0
Exp/Cntr(USF)=0,0
Exp/Cntr=0.3,0.1

Type RM Length L Ch R = 1 ,10844   ,234.3,230,217.7
XS GIS Cut Line= 3
2025452.07957862301471.2070907682025262.10744233301511.128771581
2025083.14818351301563.439939544
#Sta/Elev= 30
       0 1775.72     9.2 1774.52    22.7 1768.25    42.7 1760.33    66.2 1749.59
    72.9 1744.62      83 1738.99    97.5 1733.27   123.2 1729.48   133.2 1726.33
   144.6 1725.79   150.2 1725.06   160.1  1724.8   166.8 1725.18   170.1 1726.16
   173.5 1727.64   186.9 1735.94   191.7 1737.68   196.8  1738.4   217.5 1736.91
   231.5 1734.22   236.8 1733.71     258 1734.37   265.4 1736.55   272.2 1739.38
   289.3 1741.71     303 1745.17   340.6 1751.65   364.5 1757.15380.5695 1761.59
#Mann= 5 ,-1 , 0
       0      .1       0   144.6    .045       0   170.1      .1       0
   196.8    .016       0   217.5     .05       0
#Block Obstruct= 1 ,-1
  258.59  310.51 1766.34
Bank Sta=144.6,170.1
XS Rating Curve= 0 ,0
Exp/Cntr(USF)=0,0
Exp/Cntr=0.3,0.1

Type RM Length L Ch R = 1 ,10614   ,265.9,259,248.8
XS GIS Cut Line= 3
2025277.25014885301239.9366639862025132.70613211301352.818658011
2024937.22755709301537.284355563
#Sta/Elev= 30
       0  1791.5    10.2 1784.88    24.3 1773.92      56 1753.18    80.4 1734.21
    89.8 1728.13    95.7 1723.55    99.1 1721.75   101.8 1720.89   122.5 1720.35
     131 1722.24   138.4 1724.63   147.6 1725.06   150.6 1725.63   168.4 1732.78
   172.6 1734.04   180.9 1733.16   209.9 1732.58     232  1733.2   248.3 1732.03
   276.1 1730.16   293.5 1729.71   348.6  1729.7     362 1735.73   370.2 1741.18
   391.6 1753.79   405.9 1763.75   413.1 1767.68   434.6 1774.07452.1733 1777.49
#Mann= 5 ,-1 , 0
       0      .1       0    99.1    .045       0     131     .05       0
   248.3    .016       0   276.1     .05       0
#Block Obstruct= 2 ,-1
  149.45   183.4 1753.21   289.7  337.18 1749.79
Bank Sta=99.1,131
XS Rating Curve= 0 ,0
Exp/Cntr(USF)=0,0
Exp/Cntr=0.3,0.1

Type RM Length L Ch R = 1 ,10355   ,306.4,315.3,310.5
XS GIS Cut Line= 3
2025015.69430904301089.8862085142024941.35738614301244.066493036
2024809.20285655301508.375552215
#Sta/Elev= 30
       0 1772.65    13.4 1765.11    28.2 1751.88    35.8    1746    60.8 1730.21
    68.1 1721.51    71.7 1718.19    75.4 1716.48      79 1716.32    93.6  1716.4
   101.8 1718.23   108.1 1722.25   111.6 1723.07   133.3 1724.03   159.1 1727.45
   192.1 1728.87   203.1 1728.53   221.4 1726.75   234.2 1727.53   261.8 1727.35
   342.5 1725.91   353.5 1727.07   364.5 1732.04   375.5 1741.48   383.4 1746.77
   401.1 1760.34   407.8  1764.1   437.8 1773.95   448.8 1775.13466.6718 1780.54
#Mann= 5 ,-1 , 0
       0      .1       0    71.7    .045       0   101.8     .05       0
   234.2    .016       0   261.8     .05       0
#Block Obstruct= 2 ,-1
  127.02  171.17 1748.13  292.46  335.38 1746.97
Bank Sta=71.7,101.8
XS Rating Curve= 0 ,0
Exp/Cntr(USF)=0,0
Exp/Cntr=0.3,0.1

Type RM Length L Ch R = 1 ,10039   ,173,185.9,193.1
XS GIS Cut Line= 4
2024752.76185954301004.5364081542024685.30798506301121.548231229
2024656.39918171301183.495666974 2024575.1792104301389.987119458
#Sta/Elev= 30
       0 1745.73    17.8    1736    29.2 1730.96    44.3 1725.48    53.6 1723.49
    67.1 1719.19      86  1716.5     109 1716.28   116.3  1715.8   123.9 1716.11
   127.6 1715.69   137.7 1713.35   153.3 1711.92   156.9 1711.18   171.4 1710.64
     175 1710.74   177.2 1712.31   182.3 1717.64   184.6 1718.83   187.1 1719.62
   193.1  1720.4   222.1  1721.4   303.1 1725.55   319.3  1727.7   348.5 1733.41
   359.1 1734.23   369.7 1736.49   390.8 1742.38     419 1753.89425.3135 1755.92
#Mann= 6 ,-1 , 0
       0      .1       0   153.3    .045       0   177.2      .1       0
   193.1    .016       0   222.1     .05       0   319.3      .1       0
#XS Ineff= 2 , 0
          123.64  1717.5
Permanent Ineff=
       F       F
#Block Obstruct= 1 ,-1
  268.71  291.77 1744.97
Bank Sta=153.3,177.2
XS Rating Curve= 0 ,0
Exp/Cntr(USF)=0,0
Exp/Cntr=0.3,0.1

Type RM Length L Ch R = 1 ,9854    ,327,324.8,323.1
XS GIS Cut Line= 3
2024610.97106217300967.367946707 2024444.4012905301098.145866614
2024270.94847041301242.689883352
#Sta/Elev= 30
       0 1742.94    26.8 1729.14    47.5 1721.98    58.6 1715.99      64 1714.74
    74.6 1714.25    78.1 1712.76    82.7 1709.21    85.2 1707.42    87.4 1707.07
   101.4 1706.63   106.4 1707.12   111.8 1709.11   122.5 1714.92   129.5 1715.85
   150.5  1716.4   175.5 1714.58   233.2 1714.32   244.3 1711.36   253.2 1710.61
   279.3 1711.55   290.5  1710.6   299.8 1711.41   312.6 1710.48   320.3 1711.22
   330.5 1714.11   345.9 1717.99     393 1727.16   406.5 1731.16437.5593  1743.5
#Mann= 6 ,-1 , 0
       0      .1       0    82.7    .045       0   111.8      .1       0
   129.5    .016       0   150.5     .05       0   330.5      .1       0
#XS Ineff= 2 , 0
                          145.63         1716.76
Permanent Ineff=
       F       F
Bank Sta=82.7,111.8
XS Rating Curve= 0 ,0
Exp/Cntr(USF)=0,0
Exp/Cntr=0.3,0.1

Type RM Length L Ch R = 1 ,9529    ,210.2,206.1,205.6
XS GIS Cut Line= 3
2024392.09012253300715.4483746772024269.57186073300832.460197751
2024047.93770173301038.951650235
#Sta/Elev= 30
       0 1749.36      29 1743.32    48.4 1737.67    75.4 1728.55    79.9  1725.5
    82.3 1722.89    89.2 1714.55    93.7 1707.58    98.3 1702.55   102.8 1701.22
     121  1701.5   141.7 1700.61   147.3 1701.12   149.6 1702.16   155.9  1708.1
   161.2 1709.51   184.3 1709.75   188.8 1709.14     199 1704.33   215.7 1704.03
   233.2 1702.58   314.3 1704.65   351.6 1703.34   362.7 1705.22   372.6 1711.68
   379.4 1714.49     391 1715.28     406 1718.01   425.3 1724.05472.3379  1749.2
#Mann= 6 ,-1 , 0
       0      .1       0     121    .045       0   149.6      .1       0
   161.2    .016       0   184.3     .05       0   379.4      .1       0
#XS Ineff= 2 , 0
                          177.46         1710.18
Permanent Ineff=
       F       F
Bank Sta=121,149.6
XS Rating Curve= 0 ,0
Exp/Cntr(USF)=0,0
Exp/Cntr=0.3,0.1

Type RM Length L Ch R = 1 ,9323    ,153.1,168,151.7
Node Name=C
XS GIS Cut Line= 4
2024251.67593485 300554.385041742024178.71562163 300635.60501305
2024120.89801494300701.6822778452023925.41943992300894.407633496
#Sta/Elev= 30
       0 1716.11    12.8 1711.62    18.1 1710.64    61.4 1707.54    65.8 1706.88
    82.8 1700.04    97.1 1699.23   102.4  1698.2   107.3 1696.84     118  1696.1
   127.3 1696.22   132.2 1697.71   138.9 1699.19   152.1 1698.98   157.5 1699.53
   170.9 1703.95     184 1704.79   206.2 1704.78   220.4 1703.27   264.3 1705.41
   287.5 1705.03     320 1706.33   338.5 1706.19   347.8 1706.87   362.8 1709.84
   379.3 1711.55   416.7 1720.15   441.2 1729.39   452.2 1734.56471.4882 1742.51
#Mann= 6 ,-1 , 0
       0      .1       0   102.4    .045       0   132.2      .1       0
     184    .016       0   206.2     .05       0   379.3      .1       0
#Block Obstruct= 1 ,-1
  305.77  335.98 1726.21
Bank Sta=102.4,132.2
XS Rating Curve= 0 ,0
Exp/Cntr(USF)=0,0
Exp/Cntr=0.3,0.1

Type RM Length L Ch R = 1 ,9155    ,163.5,186.6,145.4
XS GIS Cut Line= 3
2024153.93664734300449.7627058152024014.89906933 300588.80028382
2023840.06963956300755.370055491
#Sta/Elev= 30
       0 1728.49    18.3 1717.04    45.5 1702.94    53.1 1694.81      56 1693.23
      64  1692.5    71.6 1693.13    76.3 1694.12   105.8 1695.03   124.4 1694.52
   133.6 1692.11   141.2    1694   152.2 1694.01   166.7 1695.85   178.3 1695.65
   189.3 1699.43     194 1700.21   213.1 1700.19   222.4 1699.03     236 1698.79
   313.1  1702.2   326.8 1705.66   345.4 1707.09     357 1712.27   365.1 1714.39
   376.5 1718.55   394.6 1727.12   403.4  1737.2   417.4 1748.51438.1052 1761.17
#Mann= 6 ,-1 , 0
       0      .1       0      56    .045       0    71.6      .1       0
     194    .016       0   213.1     .05       0   365.1      .1       0
Bank Sta=56,71.6
XS Rating Curve= 0 ,0
Exp/Cntr(USF)=0,0
Exp/Cntr=0.3,0.1

Type RM Length L Ch R = 1 ,8968    ,151.7,159.2,154.8
XS GIS Cut Line= 2
2024016.27567901300363.0362957712023827.68015241300594.306722553
#Sta/Elev= 30
       0 1719.16    34.9  1701.8    47.6 1696.02    54.4 1693.34    68.4 1688.83
    75.4 1688.66    81.4 1689.81    88.8 1690.13   101.1 1688.53   106.8 1687.15
   119.5 1686.31   125.2  1685.8   132.2 1685.97   136.5  1686.6   140.7 1687.59
   143.1 1688.61   144.9 1689.83   149.2 1693.87   152.4 1695.61   163.4 1696.43
   180.4 1696.01     192 1695.22   208.2 1696.87   233.8 1701.82   244.6  1705.3
   259.2 1714.95   276.2 1724.21   284.6 1729.17   292.3 1732.66298.4196 1736.16
#Mann= 5 ,-1 , 0
       0      .1       0   119.5    .045       0   136.5      .1       0
   163.4    .016       0   180.4      .1       0
Bank Sta=119.5,136.5
XS Rating Curve= 0 ,0
Exp/Cntr(USF)=0,0
Exp/Cntr=0.3,0.1

Type RM Length L Ch R = 1 ,8809    ,252.1,254,254.1
XS GIS Cut Line= 2
2023906.14690436300273.5566663622023707.91510997300491.060996311
#Sta/Elev= 30
       0 1722.63    23.4 1710.95    55.5 1693.57      66 1691.04    85.5 1689.46
   104.4 1687.06   108.8 1686.09   116.2 1682.67   119.5 1681.97   135.4 1681.68
   139.9 1681.85   143.9  1682.8   148.7 1689.55   153.4 1691.51   160.4 1691.93
   175.4 1691.66   192.6 1690.65   195.2 1692.17   197.5 1694.31   202.2 1703.41
   207.2 1718.22   209.1 1723.13   210.9 1726.84   212.1 1728.51     217 1731.96
   227.7 1737.63   233.1 1742.09   250.8 1751.12   264.2 1756.61294.2856 1767.52
#Mann= 5 ,-1 , 0
       0      .1       0   116.2    .045       0   143.9      .1       0
   160.4    .016       0   175.4      .1       0
Bank Sta=116.2,143.9
XS Rating Curve= 0 ,0
Exp/Cntr(USF)=0,0
Exp/Cntr=0.3,0.1

Type RM Length L Ch R = 1 ,8555    ,298,295.8,293.7
XS GIS Cut Line= 2
2023698.27884219300145.5319658222023464.25519604300368.542734504
#Sta/Elev= 30
       0  1700.1    17.9 1690.99      28 1687.59    36.5 1686.71    55.2 1686.47
    73.6 1687.48    91.5 1687.22    96.8 1685.62   103.8 1679.98   107.2 1677.95
   109.6 1677.32   122.3 1677.03   130.9 1677.12   133.9 1678.13   140.9 1682.07
     150 1683.29   161.8 1683.85   183.2 1682.84   192.8 1684.15   208.2 1684.09
   229.1 1684.87   231.4 1685.61   238.4  1690.5   254.6 1700.92   268.8 1712.07
   277.8 1717.15   290.9 1722.77   304.5 1726.68   313.5 1728.42323.2659 1731.75
#Mann= 6 ,-1 , 0
       0     .05       0   107.2    .045       0   133.9      .1       0
   192.8    .016       0   208.2      .5       0   238.4      .1       0
#XS Ineff= 2 , 0
                          164.85         1684.33
Permanent Ineff=
       F       F
#Block Obstruct= 2 ,-1
   75.74  100.41 1707.46  214.43  226.32 1704.35
Bank Sta=107.2,133.9
XS Rating Curve= 0 ,0
Exp/Cntr(USF)=0,0
Exp/Cntr=0.3,0.1

Type RM Length L Ch R = 1 ,8259    ,378,383.2,382
XS GIS Cut Line= 3
2023473.89146382299934.9106842882023343.11354392 300089.09096881
2023183.42682066300287.322763194
#Sta/Elev= 30
       0 1699.91    14.2 1699.06    19.2 1697.76    57.1 1681.22      71 1676.38
    97.8 1674.43   117.6 1675.71   122.3 1674.48   129.2 1671.41   149.4 1670.66
   152.5 1670.77   154.8 1671.62     158 1674.18   161.3 1675.23   188.1 1674.31
   192.1 1674.68   203.7 1677.57   224.7 1677.94   251.6 1678.08   289.5 1680.38
     296 1682.75   314.8 1693.43   323.2 1696.27   344.3  1699.5   358.7 1702.68
   376.4 1703.66   386.4 1706.08   404.4 1707.99   420.7 1710.82456.7242 1715.38
#Mann= 5 ,-1 , 0
       0      .1       0   129.2    .045       0   154.8      .1       0
   203.7    .016       0   224.7      .1       0
#XS Ineff= 2 , 0
           113.8 1677.85  169.58         1678.54
Permanent Ineff=
       F       F
Bank Sta=129.2,154.8
XS Rating Curve= 0 ,0
Exp/Cntr(USF)=0,0
Exp/Cntr=0.3,0.1

Type RM Length L Ch R = 1 ,7876    ,330.3,332,332.2
XS GIS Cut Line= 2
2023252.25730482299652.7056992272022930.13063895299948.676781121
#Sta/Elev= 30
       0 1711.11    18.5 1711.04    32.3 1709.28    48.7 1704.68      65 1697.59
    85.9 1690.22    90.9 1687.08   103.5 1671.41   110.3 1667.68   129.7 1665.79
   153.9 1665.69   178.2 1667.08   190.4 1663.05   208.9 1661.63   218.2 1662.81
   234.5 1665.92   294.6 1666.87   309.1  1673.4   320.4 1674.58   333.4 1675.25
   341.3 1674.51   345.9 1675.42   357.5 1682.39   367.3  1685.3   386.7 1694.26
   390.1 1698.23     397 1712.12   401.2 1717.72   425.5 1736.79437.4522 1744.98
#Mann= 5 ,-1 , 0
       0     .05       0   190.4    .045       0   218.2     .05       0
   320.4    .016       0   333.4      .1       0
#XS Ineff= 2 , 0
             150 1668.79  237.75         1668.79
Permanent Ineff=
       F       F
#Block Obstruct= 1 ,-1
  241.77  254.02 1686.16
Bank Sta=190.4,218.2
XS Rating Curve= 0 ,0
Exp/Cntr(USF)=0,0
Exp/Cntr=0.3,0.1

Type RM Length L Ch R = 1 ,7544    ,300.9,321.7,332.9
XS GIS Cut Line= 2
2023054.02551044299399.4095175142022661.69175072299733.925670538
#Sta/Elev= 30
       0  1692.1     6.4 1689.89      25 1680.43      39 1670.74    45.3 1667.42
      53 1665.94    63.9 1664.93    72.5 1663.07   136.8 1659.98   222.2 1659.35
   227.3 1658.73   232.4 1656.62   237.4 1654.99     245 1654.51   253.1 1654.74
   260.1 1656.45   296.7 1659.23   308.2 1661.97   318.3  1668.2   322.6 1669.89
   332.3  1671.2   357.1 1672.63   361.4 1675.26   365.7 1683.18     370 1692.97
   374.1 1699.64   391.6 1711.24   443.3 1726.87   475.1 1734.24 515.584 1740.82
#Mann= 5 ,-1 , 0
       0      .1       0   232.4    .045       0   260.1     .05       0
   332.3    .016       0   357.1      .1       0
#XS Ineff= 2 , 0
          199.44 1663.37  283.61         1662.31
Permanent Ineff=
       F       F
Bank Sta=232.4,260.1
XS Rating Curve= 0 ,0
Exp/Cntr(USF)=0,0
Exp/Cntr=0.5,0.3

Type RM Length L Ch R = 1 ,7222    ,52.7,52.5,52.4
XS GIS Cut Line= 5
2023024.27532081299347.123449789 2022720.9806754299310.326672957
2022649.61722942  299311.44172682022547.03227583 299318.13204986
2022428.83656843299349.353557476
#Sta/Elev= 30
       0 1690.95    45.4 1673.01      62 1667.29    78.5 1662.94    85.1 1660.53
   131.4 1660.24   147.9  1662.6   158.8 1662.77   180.9 1661.74   220.6 1657.53
   306.5 1656.13   316.4 1655.32   326.2 1652.44   342.4 1649.97   352.5 1649.54
     359 1650.23   361.8 1652.38   368.9 1659.73   374.7 1662.54   378.7 1664.02
   388.6 1664.14   411.3 1665.11   424.7  1664.8   434.6 1666.82     451 1674.04
   541.7 1706.86   551.9 1709.04   565.6 1709.77   582.5 1710.26601.9435 1709.62
#Mann= 5 ,-1 , 0
       0     .05       0   326.2    .045       0   361.8     .05       0
   388.6    .016       0   411.3     .05       0
#XS Ineff= 3 ,-1
       0     280    1662     280     298  1656.7   386.5     500 1661.88
Permanent Ineff=
       F       F       F
#Block Obstruct= 2 ,-1
  121.61  179.21 1681.81   564.5  601.94  1729.7
Bank Sta=326.2,361.8
XS Rating Curve= 0 ,0
Exp/Cntr(USF)=0,0
Exp/Cntr=0.5,0.3

Type RM Length L Ch R = 3 ,7183    ,,,
BEGIN DESCRIPTION:
Private Driveway
Survey ID: LIC110
END DESCRIPTION:
Bridge Culvert--1,0,-1,-1, 0
Deck Dist Width WeirC Skew NumUp NumDn MinLoCord MaxHiCord MaxSubmerge Is_Ogee
23,12,2.6,0, 10, 10, , , 0.98, 0, 0,0,,
     260     307     312   316.5   316.5     344     360   363.5   363.5     376
1656.3551657.2631658.197 1659.06 1659.061659.9521661.3461661.3461661.3461662.017
                                 1657.561658.4521659.8461659.846
     260     307     312   316.5   316.5     344     360   363.5   363.5     376
1656.3551657.2631658.197 1659.06 1659.061659.9521661.3461661.3461661.3461662.017
                                 1657.561658.4521659.8461659.846
Pier Skew, UpSta & Num, DnSta & Num=  ,330, 2 ,330, 2 , 0 , 0 , 0 ,,
       2       2
       0    1659
       2       2
       0    1659
BR Coef=-1 , 1 , 0 ,1.25, 0 ,,,0.8,0,2,0,
WSPro=,,,, 1 ,,,, 0 ,,,, 0 ,,,,-1 ,-1 ,-1 , 0 , 0 , 0 , 0 , 0
BC Design=,, 0 ,, 0 ,,,,,,
BC Use User HTab Curves=0
BC User HTab FreeFlow(D)= 0

Type RM Length L Ch R = 1 ,7170    ,230.3,220,205.8
XS GIS Cut Line= 5
2023024.27532081299294.715919149 2022720.9806754299257.919142316
2022649.61722942 299259.034196162022547.03227583 299265.72451922
2022428.83656843299296.946026836
#Sta/Elev= 30
       0 1702.16    12.4  1699.1    29.1 1691.64    58.7 1680.85   101.6 1663.27
   124.8 1657.51   141.1 1658.54   158.8 1658.39   208.9 1655.75   237.1 1655.76
   280.1 1653.88   316.4 1654.37   326.2 1652.75   326.3 1652.73   349.2 1649.41
   361.7  1651.5   364.9 1653.08   372.1 1660.85   375.4 1661.91     382 1660.69
   388.6 1660.69   407.9 1662.73   433.3 1663.88   444.5 1664.09   457.6  1667.5
   493.1 1670.73     535 1689.15   565.5  1699.4   582.5  1703.5601.9435 1702.58
#Mann= 6 ,-1 , 0
       0     .05       0   326.2    .045       0   326.3    .045       0
   364.9     .05       0   407.9    .016       0   433.3     .05       0
#XS Ineff= 3 ,-1
       0     300    1660     300     309  1655.1 370.167     500 1659.77
Permanent Ineff=
       F       F       F
#Block Obstruct= 1 ,-1
  216.78  268.54 1675.71
Bank Sta=326.3,364.9
XS Rating Curve= 0 ,0
Exp/Cntr(USF)=0,0
Exp/Cntr=0.5,0.3

Type RM Length L Ch R = 1 ,6950    ,301.9,313.8,276.6
XS GIS Cut Line= 3
 2022859.9235451298986.4266125462022620.39346022299062.140145124
2022292.76035562299152.996384217
#Sta/Elev= 30
       0 1693.89    12.6    1694    19.5  1693.2    36.7 1684.23    53.9 1677.33
    64.2 1675.21     102 1671.08   147.7 1652.84   152.9 1651.67     164 1651.41
   174.3 1647.14     179  1646.2   186.9  1645.9   202.6 1647.36   218.3    1649
   253.4 1651.17   294.3 1652.49   310.9 1657.32   318.1 1658.26   334.1 1658.54
   345.3 1658.29   355.6 1661.09     376 1664.53     393 1665.06   413.4 1668.35
   433.9  1668.7   443.9 1670.37   481.6 1673.92     506 1678.53 591.209 1698.23
#Mann= 6 ,-1 , 0
       0    .016       0    19.5     .05       0   174.3    .045       0
   202.6     .05       0   318.1    .016       0   334.1     .05       0
#Block Obstruct= 3 ,-1
  399.61  413.61 1688.35  418.51  427.36 1688.37  438.09  454.77 1691.26
Bank Sta=174.3,202.6
XS Rating Curve= 0 ,0
Exp/Cntr(USF)=0,0
Exp/Cntr=0.3,0.1

Type RM Length L Ch R = 1 ,6636    ,307,320.4,300.2
XS GIS Cut Line= 3
2022711.24969932298757.9094051312022566.70568258 298817.10362151
2022243.20240702298914.842909019
#Sta/Elev= 30
       0  1680.5    36.7 1662.53    54.9 1653.04    61.5 1650.14      70 1647.37
    82.7 1645.37    90.1 1641.74    93.4 1640.35    96.9 1639.77   112.7 1641.88
   125.3 1643.94   181.2 1644.87   201.7 1648.43   221.3 1649.25   239.7 1651.51
   246.3 1651.92     260 1651.94   270.3 1651.35   287.1 1654.45   314.8 1657.65
   325.1 1659.22   337.1 1661.19   359.4 1665.63   391.2 1668.73   407.4  1671.2
   438.2 1677.06   445.1 1677.92   458.8 1680.52   476.6 1685.02494.1409 1690.65
#Mann= 5 ,-1 , 0
       0     .05       0    90.1    .045       0   112.7     .05       0
   239.7    .016       0     260     .05       0
#Block Obstruct= 1 ,-1
  346.88  391.57 1688.78
Bank Sta=90.1,112.7
XS Rating Curve= 0 ,0
Exp/Cntr(USF)=0,0
Exp/Cntr=0.3,0.1

Type RM Length L Ch R = 1 ,6316    ,343,343.5,345.8
Node Name=B
XS GIS Cut Line= 3
2022652.05548294298517.0027105662022462.08334665298567.937268846
2022009.17876087298678.066043504
#Sta/Elev= 30
       0 1681.75    21.4 1682.09    31.6 1678.91    86.3 1652.11      97 1645.75
   106.3 1641.75   113.1 1637.09   116.5 1635.38   123.3 1634.88   130.1 1635.17
   134.5 1636.72   140.3  1640.2   143.7 1640.91   187.4 1641.97   209.7  1643.9
     225 1644.31   236.9  1645.7   248.7 1644.36     264 1645.02   349.9 1643.67
     404 1647.64   444.5 1653.63   507.5 1667.46   528.9 1675.79   569.4 1688.93
   586.3 1693.35   613.3 1703.81   626.8 1707.81   647.1 1711.25662.7836 1715.88
#Mann= 6 ,-1 , 0
       0    .016       0    21.4     .05       0   113.1    .045       0
   134.5     .05       0   209.7    .016       0     225     .05       0
#Block Obstruct= 1 ,-1
  353.79  414.36 1669.13
Bank Sta=113.1,134.5
XS Rating Curve= 0 ,0
Exp/Cntr(USF)=0,0
Exp/Cntr=0.3,0.1

Type RM Length L Ch R = 1 ,5972    ,295.5,297.1,294.2
XS GIS Cut Line= 4
2022557.06941479298214.1485802572022384.99320439298255.446870754
2022329.92881706298267.8363579032021843.98559888298397.237668126
#Sta/Elev= 30
       0 1674.53      45 1674.44    55.1 1672.61    71.6 1664.89   109.1 1639.37
   119.3 1632.94     126  1629.9   132.8 1627.45   142.9 1626.85   149.6 1627.63
   153.9 1629.95   159.7 1634.62   173.7 1638.24   197.6 1637.26   210.2 1638.23
     217 1636.86   243.9 1635.86   267.7 1636.45   284.7 1635.58   297.7 1638.38
   322.1 1638.17     488 1637.29   522.4 1638.13   541.7 1639.84   573.3 1645.77
   627.6 1659.43   643.5 1666.79   691.8 1685.28   715.8 1696.93736.2809 1705.37
#Mann= 6 ,-1 , 0
       0    .016       0      45     .05       0     126    .045       0
   153.9     .05       0   297.7    .016       0   322.1     .05       0
#Block Obstruct= 2 ,-1
   386.9   424.8 1658.12  435.84  471.91 1658.03
Bank Sta=126,153.9
XS Rating Curve= 0 ,0
Exp/Cntr(USF)=0,0
Exp/Cntr=0.3,0.1

Type RM Length L Ch R = 1 ,5675    ,277.5,279.3,281.7
XS GIS Cut Line= 3
2022409.77217869297964.9822275932022111.04787743298059.968295736
2021788.92121156298310.511258083
#Sta/Elev= 30
       0 1639.59     9.4 1638.19    55.9 1637.95    70.4 1636.26    77.4 1635.11
   101.4 1626.71   111.7 1625.87   120.9 1622.45   132.4 1620.19   146.1 1620.38
   149.6 1621.28     153 1623.72   156.5  1626.3   160.9 1627.93   187.5 1629.98
   205.3 1630.09     215 1628.96   221.9 1626.07   225.3  1625.4     246 1625.19
   331.3 1631.04   402.4 1633.42   565.8 1643.44   597.5 1646.86   630.5 1653.16
   635.2  1654.8   655.9 1665.41   693.3 1677.94     710 1680.76721.5521  1681.3
#Mann= 5 ,-1 , 0
       0     .05       0   120.9    .045       0     153     .05       0
   187.5    .016       0   205.3     .05       0
#XS Ineff= 2 , 0
                          203.72         1630.55
Permanent Ineff=
       F       F
Bank Sta=120.9,153
XS Rating Curve= 0 ,0
Exp/Cntr(USF)=0,0
Exp/Cntr=0.3,0.1
